--- SOVERNRN.prj (project) ---

Proj Title=SOVERNRN
Current Plan=p01
Default Exp/Contr=0,0
English Units
Geom File=g01
Flow File=f01
Plan File=p01
BEGIN DESCRIPTION:
END DESCRIPTION:
DSS Export Rating Curves= 0
DSS Export Rating Curve Sorted= 0
DSS Export Volume Flow Curves= 0
DXF OffsetX= 0
DXF OffsetY= 0
DXF ScaleX= 0
DXF ScaleY= 0

--- SOVERNRN.p01 (plan) ---

Plan Title=Floodplain
Program Version=4.00
Geom File=g01
Flow File=f01
K Sum by GR=0
Std Step Tol=0.01
Critical Tol=0.01
Num of Std Step Trials=20
Max Error Tol=0.3
Flow Tol Ratio=0.001
Split Flow NTrial=30
Split Flow Tol=0.02
Split Flow Ratio=0.02
Log Output Level=0
Friction Slope Method=1
Unsteady Friction Slope Method=2
Unsteady Bridges Friction Slope Method=1
Global Log Level=0
CheckData=False
Run HTab=0
Run UNet=0
Run PostProcess=0
UNET Theta=0
UNET Theta Warmup=0
UNET ZTol=0
UNET ZSATol=0
UNET MxIter=0
UNET MaxInSteps=0
UNET DtIC=0
UNET DtMin=0
UNET MaxCRTS=0
UNET WFStab=0
UNET SFStab=0
UNET WFX=0
UNET SFX=0
UNET DSS MLevel=0
UNET DZMax Abort=0
UNET Convert EG Bridges=0
UNET Use Existing IB Tables=0
UNET Froude Limit=0
UNET Froude Power=0
Write IC File=0
Echo Input=False
Echo Output=False
Write Detailed=0

--- SOVERNRN.f01 (steady flow) ---

Flow Title=NFF Regression Equation
Program Version=4.00
Number of Profiles=1
Profile Names=P100yr
River Rch & RM=SOVERNRN,Main      ,18070.8
519.0760
River Rch & RM=SOVERNRN,Main      ,13951
578.2698
River Rch & RM=SOVERNRN,Main      ,11972.5
644.5480
River Rch & RM=SOVERNRN,Main      ,11708.6
686.1772
River Rch & RM=SOVERNRN,Main      ,8289.4
727.7333
River Rch & RM=SOVERNRN,Main      ,7873.4
897.4097
River Rch & RM=SOVERNRN,Main      ,5453.5
933.2023
River Rch & RM=SOVERNRN,Main      ,4662.9
1056.867
River Rch & RM=SOVERNRN,Main      ,281.2
1140.819
Boundary for River Rch & Prof#=SOVERNRN,Main      ,1
Up Type=0
Dn Type=3
Dn Slope=0.128363

--- SOVERNRN.g01 (geometry) ---

Geom Title=USGS 10m DEM
Program Version=4.10

River Reach=SOVERNRN        ,Main
Reach XY= 30
     1915225.798      396023.719     1915072.369      396211.653
     1914672.412       396265.69     1914392.464      396988.889
     1914108.176      397090.885     1914006.158      397358.014
     1912242.942       398577.43     1911843.636      399265.364
     1912138.318      399483.354      1912131.18      400130.165
     1911828.445       400255.49     1911814.255      400626.554
      1911435.65      401181.597     1911105.789      401246.701
     1910705.026      401714.397      1910812.82      402176.063
     1909992.485      402382.021     1909833.003      402530.881
     1909894.852      402722.938     1909553.202      402951.906
     1909609.587      403208.661     1909964.296      403100.542
     1910479.704      403644.705     1910157.438      404432.465
     1910405.919      404779.145     1910173.714      406050.846
     1910544.808      406795.204      1910801.97      406988.889
     1910718.419       407331.77     1911030.486       408421.24

Type RM Length L Ch R = 1 ,18070.8 ,340,365.6,390.4
XS GIS Cut Line= 3
     1914945.785      395882.118     1915123.736      396048.133
     1915330.984       396238.02
#Sta/Elev= 30
       0 1907.73    48.7 1898.64    58.4  1897.1    68.1 1895.77    77.9 1894.62
    87.6  1893.7   126.6 1890.67   136.3 1889.97     146 1889.42   155.8  1889.5
   165.5  1889.9   175.2 1890.09   204.4 1889.26   253.1  1887.4   262.8 1886.61
   272.4  1884.1   282.1 1881.23   291.8 1879.55   302.5 1880.26   330.6 1883.32
   369.4 1887.25   379.1 1888.42   388.8 1891.12   398.4  1895.4   417.8 1906.05
   427.5 1911.04   437.2  1915.5   456.6 1923.91   505.1 1945.34   524.4 1953.99
#Mann= 3 , 0 , 0
       0      .1       0   282.1    .045       0   302.5      .1       0
Bank Sta=282.1,302.5
XS Rating Curve= 0 ,0
Exp/Cntr=0.3,0.1

Type RM Length L Ch R = 1 ,17705.3 ,421.6,379.1,336
XS GIS Cut Line= 4
     1914862.234      396030.772     1914891.531      396205.468
     1914877.425      396290.104     1914969.656      396424.652
#Sta/Elev= 29
       0 1900.17    39.4 1894.67    68.9 1890.69    98.4 1886.21   108.2 1884.82
   118.1 1883.91   127.9 1883.43   137.8 1883.24   147.6  1883.3   167.3 1883.76
   177.1  1883.8   186.7 1883.02   196.2 1880.75   205.2 1877.21   215.3 1873.82
   224.8 1874.05   225.2 1874.21   243.9 1881.48   253.4 1883.24   272.5 1885.17
   282.1 1886.43   310.9 1890.49   339.7  1894.3   368.5 1897.99   378.1 1898.98
   397.3 1900.65   406.9 1902.07   416.5    1904   426.1 1906.28
#Mann= 3 , 0 , 0
       0      .1       0   205.2    .045       0   225.2      .1       0
Bank Sta=205.2,225.2
XS Rating Curve= 0 ,0
Exp/Cntr=0.3,0.1

Type RM Length L Ch R = 1 ,17326.1 ,220.6,235.2,249.5
XS GIS Cut Line= 3
     1914469.439      396373.654     1914600.733      396402.951
     1914789.535      396408.376
#Sta/Elev= 26
       0 1913.03     9.6 1911.52    19.2 1909.79      48 1904.29    57.6 1902.29
    76.9 1897.66    86.5 1895.58    96.1 1893.75   115.3 1890.51   124.9 1887.96
   134.5 1882.33     144 1872.05   148.5 1868.13   153.4 1863.86   162.8 1863.81
   168.5 1866.75   172.3 1868.71   181.7 1873.32   191.2 1874.77   210.1 1875.91
   219.5 1876.63     229 1877.43   247.8 1879.17   257.3 1880.14   285.6 1883.29
   323.4 1887.72
#Mann= 3 , 0 , 0
       0      .1       0   148.5    .045       0   168.5      .1       0
Bank Sta=148.5,168.5
XS Rating Curve= 0 ,0
Exp/Cntr=0.3,0.1

Type RM Length L Ch R = 1 ,17091   ,270.2,266.1,262.1
XS GIS Cut Line= 2
     1914427.122      396539.127     1914649.561      396694.292
#Sta/Elev= 19
       0 1886.76    58.1 1882.64    87.2 1880.66    96.9 1879.17   106.6 1874.48
   116.2 1866.91   123.5 1862.32   125.9 1860.81   135.6 1860.33   143.5 1862.39
   145.3 1862.86     155  1867.2   164.7 1871.76   174.4 1876.02     184  1879.6
   193.7  1881.8   203.4 1882.93   242.2 1885.91   271.2 1887.98
#Mann= 3 , 0 , 0
       0      .1       0   123.5    .045       0   143.5      .1       0
Bank Sta=123.5,143.5
XS Rating Curve= 0 ,0
Exp/Cntr=0.3,0.1

Type RM Length L Ch R = 1 ,16824.8 ,228.3,248.1,266.9
XS GIS Cut Line= 3
     1914273.128      396690.603     1914355.594      396817.556
     1914549.821      396910.872
#Sta/Elev= 28
       0  1871.8     9.5 1870.77    18.9  1869.9    28.4  1869.2    47.3 1868.05
    94.6 1865.47   113.5 1864.21     123 1863.49   132.5 1862.64   141.9 1861.57
   151.4 1859.74   161.2 1856.96     171 1853.52   180.8 1852.13   193.5  1853.4
   200.4 1854.11     220 1855.75   229.7 1856.76   239.5 1858.57   249.3 1861.79
   259.1 1866.41   268.9 1871.64   278.7 1876.73   288.5 1879.75   298.3  1881.2
   337.5 1885.52   357.1 1887.56   366.9 1888.92
#Mann= 3 , 0 , 0
       0      .1       0     171    .045       0   193.5      .1       0
Bank Sta=171,193.5
XS Rating Curve= 0 ,0
Exp/Cntr=0.3,0.1

Type RM Length L Ch R = 1 ,16576.7 ,165.5,168.6,171.5
XS GIS Cut Line= 3
     1914248.953      396848.589     1914320.568      397029.579
     1914429.943      397176.714
#Sta/Elev= 29
       0 1859.87     9.7 1858.13    19.5 1855.93    29.2 1854.63    38.9 1853.93
    58.4  1852.8   136.2  1848.7     146 1847.58   155.7 1844.88   165.4 1842.74
   175.2 1843.18   177.4 1844.05   184.9 1847.02   204.3 1858.97   213.9 1864.36
   223.6 1869.65   233.2 1874.52   242.9 1878.11   252.5 1880.64   262.2 1881.69
   271.8 1882.02   291.1 1882.93   300.8 1883.59   310.4  1884.4   320.1 1885.35
   329.7 1886.57   339.4 1888.25   368.3 1893.89     378 1895.63
#Mann= 3 , 0 , 0
       0      .1       0   155.7    .045       0   177.4      .1       0
Bank Sta=155.7,177.4
XS Rating Curve= 0 ,0
Exp/Cntr=0.3,0.1

Type RM Length L Ch R = 1 ,16408.1 ,318.1,307.5,296.6
XS GIS Cut Line= 3
     1914111.284      396907.147     1914159.027      397085.098
     1914269.704      397215.306
#Sta/Elev= 27
       0 1858.15     9.7  1857.3    19.4 1856.72    38.8 1856.16    48.5 1855.75
    58.2 1855.11    67.9  1854.2      97 1851.16   116.4 1848.94   126.1 1847.15
   135.8 1843.72   145.5 1839.83   148.8 1839.26   155.2 1838.14   164.8 1838.17
   174.6  1838.4   193.7 1838.86   241.2 1840.29   250.7 1840.87   260.2 1842.76
   269.7 1846.52   288.7 1855.82   307.7 1864.96   317.2 1869.14   326.6 1871.91
   336.2 1873.45   355.1 1875.54
#Mann= 3 , 0 , 0
       0      .1       0   148.8    .045       0   174.6      .1       0
Bank Sta=148.8,174.6
XS Rating Curve= 0 ,0
Exp/Cntr=0.3,0.1

Type RM Length L Ch R = 1 ,16100.6 ,381.4,372.7,371
XS GIS Cut Line= 4
     1914021.089      396963.823     1913985.932      397211.219
     1914008.068      397295.855     1914147.391      397462.521
#Sta/Elev= 30
       0  1854.4    57.7 1851.59    76.9 1849.16    96.1 1845.21   105.7 1843.96
   115.3 1843.76   124.9 1844.19   182.6 1847.56     221 1847.37   240.3 1846.68
   249.9 1845.53     279 1839.98   298.5 1836.73   317.9  1834.9   356.2 1832.55
     370  1830.2   384.6  1828.1     394 1828.37   403.5 1829.63   422.4 1833.16
   431.8 1835.49   441.3 1840.42   460.2 1855.95   469.6 1860.92     479  1864.3
   497.9  1869.6   507.4 1871.37   526.3 1872.93   535.7 1874.76   554.6 1880.27
#Mann= 3 , 0 , 0
       0      .1       0     370    .045       0     394      .1       0
Bank Sta=370,394
XS Rating Curve= 0 ,0
Exp/Cntr=0.3,0.1

Type RM Length L Ch R = 1 ,15727.9 ,384.2,394.5,394.8
XS GIS Cut Line= 3
     1913694.266      397194.292     1913695.568      397476.844
     1913842.703      397639.605
#Sta/Elev= 30
       0 1839.64      39 1838.69      78 1837.55   136.4 1835.28   165.6 1833.99
   204.6 1832.56   224.1 1832.03   233.8 1831.56   243.6 1830.53   292.1    1824
   301.6 1822.46   311.2 1820.73  316.911820.057   320.7 1819.61   330.2 1819.89
   339.8 1821.11   342.9 1821.66   349.3  1822.8   358.9 1824.15   368.4 1825.27
     378 1826.13     397 1827.22   406.6 1828.16   416.1 1829.42   425.6 1831.04
   444.7 1834.48   454.3 1836.34   473.3 1840.34   482.9 1842.47     502  1846.9
#Mann= 3 , 0 , 0
       0      .1       0  316.91    .045       0   342.9      .1       0
Bank Sta=316.91,342.9
XS Rating Curve= 0 ,0
Exp/Cntr=0.3,0.1

Type RM Length L Ch R = 1 ,15333.5 ,366.2,369.6,372.7
XS GIS Cut Line= 3
     1913342.703      397416.948     1913457.286      397713.823
     1913599.214      397860.959
#Sta/Elev= 30
       0 1830.34    19.3 1829.05    28.9 1828.66    48.2 1828.39    77.1 1828.29
   154.3 1827.32   183.2 1826.82   212.2  1826.2   221.8 1825.88   231.4 1825.11
   241.1 1823.59   260.4 1819.87     270 1818.27   279.6 1817.17   289.3 1816.51
   298.9 1816.06   347.4 1814.18   357.2 1813.11   366.9 1811.33   376.6 1810.22
   386.4 1811.84   388.2 1812.86   396.1 1817.31   405.8 1824.34   415.6 1830.97
   425.3 1835.43     435 1838.24   464.2 1843.73   503.2 1851.39   522.6 1855.04
#Mann= 3 , 0 , 0
       0      .1       0   366.9    .045       0   388.2      .1       0
Bank Sta=366.9,388.2
XS Rating Curve= 0 ,0
Exp/Cntr=0.3,0.1

Type RM Length L Ch R = 1 ,14963.8 ,334.8,328.3,321.3
XS GIS Cut Line= 4
     1913045.398      397555.671     1913139.426      397853.198
     1913187.755       397942.99     1913317.964      398121.376
#Sta/Elev= 26
       0  1823.7    48.8 1821.63     156 1816.86   204.8 1814.88   224.3 1814.35
   292.5 1812.96   302.3 1812.33     312  1810.5   321.3 1807.81   330.6    1806
   339.8  1805.3   349.1 1805.12   433.2 1804.09   442.8 1803.41   452.4 1802.32
     462 1801.93   468.2 1803.19   471.6 1803.88   481.2 1810.39   490.8 1817.93
   500.4 1823.54     510 1826.42   519.6 1828.02   548.4 1832.38     606 1841.98
   634.9 1846.57
#Mann= 3 , 0 , 0
       0      .1       0   442.8    .045       0   468.2      .1       0
Bank Sta=442.8,468.2
XS Rating Curve= 0 ,0
Exp/Cntr=0.3,0.1

Type RM Length L Ch R = 1 ,14635.6 ,210.9,229.1,247.2
XS GIS Cut Line= 3
     1912747.651      397815.386     1912926.036      398069.292
     1913121.349      398226.844
#Sta/Elev= 28
       0 1812.76     9.7 1810.24    19.4 1808.08    29.1 1806.61    38.8 1805.79
    58.2 1805.13    87.3 1804.37   155.2 1803.08   174.6 1802.59   193.9 1801.98
   232.7 1800.33   310.3 1795.81     320 1795.02   329.6 1792.57   339.3 1789.19
   348.9 1787.24   358.6 1788.29   361.5 1789.35   368.2 1791.81   377.9 1794.57
   387.5 1795.76   397.2  1797.4   406.8 1800.41   416.5 1803.92   426.1 1806.64
   435.8 1808.45   474.4 1814.39   561.2 1828.56
#Mann= 3 , 0 , 0
       0      .1       0   339.3    .045       0   361.5      .1       0
Bank Sta=339.3,361.5
XS Rating Curve= 0 ,0
Exp/Cntr=0.3,0.1

Type RM Length L Ch R = 1 ,14406.5 ,467.8,455.5,442.4
XS GIS Cut Line= 4
     1912706.505      397885.264     1912752.078      398114.431
     1912769.005      398209.483     1912918.224      398364.865
#Sta/Elev= 30
       0 1808.02    19.5 1805.46    29.2 1804.42    38.9 1803.79    77.9 1802.78
   107.1 1802.23   116.8 1801.57   126.6 1800.59   175.2  1795.1     253 1787.16
   262.6 1785.82   272.3 1783.84   281.9 1781.61   291.6 1780.56   301.2  1781.6
     303 1782.04   310.9 1783.99   320.6 1785.74     340 1785.69   349.8 1786.41
   359.6 1787.91   369.4 1790.27     389 1796.35   398.8 1799.03   408.5 1800.62
   418.3 1801.44   447.7 1803.18   467.3 1804.83   506.5 1809.08   545.6 1813.52
#Mann= 3 , 0 , 0
       0      .1       0   281.9    .045       0     303      .1       0
Bank Sta=281.9,303
XS Rating Curve= 0 ,0
Exp/Cntr=0.3,0.1

Type RM Length L Ch R = 1 ,13951   ,217.8,225.2,232
XS GIS Cut Line= 4
     1912389.578      398163.042     1912496.349      398469.032
     1912551.036      398535.438     1912644.786      398595.334
#Sta/Elev= 29
       0 1785.13    19.6 1783.47    39.3 1781.93    68.7  1780.1    98.2 1778.57
   127.7  1777.4   186.6 1775.47   235.7 1773.63   245.5 1773.38   304.4  1773.3
   333.6 1772.94   343.2 1771.93   352.8  1769.9   362.3 1768.94   371.9  1769.5
   381.4 1770.62     391 1771.81   400.6 1773.67   410.1 1776.22   419.4 1779.08
   428.6  1782.1   437.9 1785.03   447.2 1787.69   465.7 1793.47     475 1796.16
   484.3 1798.42   493.6 1800.31   512.1 1803.54   521.4 1805.06
#Mann= 3 , 0 , 0
       0      .1       0   352.8    .045       0   381.4      .1       0
Bank Sta=352.8,381.4
XS Rating Curve= 0 ,0
Exp/Cntr=0.3,0.1

Type RM Length L Ch R = 1 ,13725.8 ,461.6,454.5,447.3
XS GIS Cut Line= 3
     1912192.964      398252.886     1912333.589      398574.501
     1912527.599      398746.376
#Sta/Elev= 25
       0 1780.35      39 1778.71     117 1776.16   165.8 1774.26     234 1771.81
     273 1770.29   282.8 1769.71   292.5 1768.09   302.3 1765.44     312 1764.39
   322.5 1765.52   331.5 1767.06   341.3 1768.03     351 1768.39   389.4 1768.88
     399 1769.11   408.6 1769.52   418.2 1770.12   437.4  1771.6   466.2 1773.64
   475.8 1774.44   485.4 1775.13     591 1780.02   600.6  1780.9   610.2 1783.39
#Mann= 3 , 0 , 0
       0      .1       0   302.3    .045       0   322.5      .1       0
Bank Sta=302.3,322.5
XS Rating Curve= 0 ,0
Exp/Cntr=0.3,0.1

Type RM Length L Ch R = 1 ,13271.3 ,356,345.2,334.3
XS GIS Cut Line= 4
     1911706.857      398545.254     1912021.093      398824.768
     1912073.176      398887.268     1912476.818      398979.448
#Sta/Elev= 30
       0 1790.07    29.3 1789.45    58.7 1787.52    68.5  1786.2    97.8 1779.58
   117.4 1775.88   136.9 1773.64   156.5  1772.8   166.3 1771.89     176 1769.88
   195.6 1764.24   205.4 1763.66   332.5 1762.02   381.4  1760.8   429.6 1758.12
   438.6 1756.74   447.7 1754.56   456.7 1753.89   465.8 1754.44   469.6 1755.09
   483.8 1757.03   492.9 1757.25   627.1 1756.62   675.2 1758.36     733 1758.71
   781.2 1762.06   819.7  1765.7   877.4 1771.88   887.1 1773.31     916 1779.77
#Mann= 3 , 0 , 0
       0      .1       0   447.7    .045       0   469.6      .1       0
#XS Ineff= 2 , 0
                          493.07         1757.29
Permanent Ineff=
       F       F
Bank Sta=447.7,469.6
XS Rating Curve= 0 ,0
Exp/Cntr=0.3,0.1

Type RM Length L Ch R = 1 ,12926   ,525.2,504.1,482.5
XS GIS Cut Line= 4
     1911420.398      399251.852     1911841.401      399133.094
     1911936.887      399176.497      1912355.29      399087.955
#Sta/Elev= 30
       0 1771.78   106.9 1765.07   145.8 1762.22   155.5  1761.2   165.2 1759.83
   223.6    1751   233.3 1750.58   291.6 1750.08     350 1748.89   398.6 1749.48
     447 1749.35   456.5 1748.92     466 1747.34     473 1745.77   475.6 1745.19
   485.1 1744.21   494.6 1745.24   504.2 1747.55   513.7 1748.88   542.3 1749.12
   610.4 1751.37   649.2 1751.94   668.7 1751.95   688.1 1751.78   765.9 1750.17
   824.2  1750.7   833.9 1750.98   863.1 1752.58   950.6 1755.93     970 1757.28
#Mann= 3 , 0 , 0
       0      .1       0     473    .045       0   494.6      .1       0
Bank Sta=473,494.6
XS Rating Curve= 0 ,0
Exp/Cntr=0.3,0.1

Type RM Length L Ch R = 1 ,12421.9 ,439.1,449.4,459.2
XS GIS Cut Line= 4
      1911663.28      399685.879     1912064.496      399512.268
     1912199.912      399454.977     1912370.915      399200.803
#Sta/Elev= 30
       0 1756.89    19.4 1754.36      68 1748.67    97.2  1744.5   106.9 1743.47
   116.6 1743.02   155.4 1742.73   223.4 1740.25   252.6 1739.67   291.4 1739.98
   369.2 1742.44   388.6 1742.58   417.7 1742.24     447 1741.25   486.2 1739.09
     496 1737.66   505.8 1734.77   515.6 1732.39   525.4 1732.14   535.2 1734.47
     545 1737.18   554.8 1738.36   603.4 1738.92   632.1 1739.94   708.7 1743.79
   804.4 1749.18   823.5 1750.06   852.2    1751   861.8 1751.55   890.6 1754.25
#Mann= 3 , 0 , 0
       0      .1       0   505.8    .045       0   535.2      .1       0
Bank Sta=505.8,535.2
XS Rating Curve= 0 ,0
Exp/Cntr=0.3,0.1

Type RM Length L Ch R = 1 ,11972.5 ,239.3,264,289.1
XS GIS Cut Line= 4
     1911723.345      399864.865     1912103.554      399925.629
     1912204.248      399925.629     1912633.068      399975.976
#Sta/Elev= 30
       0 1764.05    19.2 1758.31    28.9 1755.01    67.4 1739.49      77 1736.52
    86.6  1734.7   115.5 1731.48   134.8 1730.22   259.9 1729.29   412.5 1727.25
   421.6 1726.61   430.8 1724.65     440 1722.93   449.1 1723.05   458.3 1725.94
   467.4 1728.18   476.6 1728.74   495.5 1728.59   515.2 1728.01     525 1727.36
   564.2 1723.52     574 1723.29   583.9 1724.81   603.5 1730.61   652.6 1737.81
     682 1740.69   760.5 1744.52   780.1 1746.08   819.4 1750.34   917.5  1763.9
#Mann= 3 , 0 , 0
       0      .1       0   430.8    .045       0   458.3      .1       0
#XS Ineff= 2 , 0
                          478.18         1728.61
Permanent Ineff=
       F       F
Bank Sta=430.8,458.3
XS Rating Curve= 0 ,0
Exp/Cntr=0.3,0.1

Type RM Length L Ch R = 1 ,11708.6 ,377.6,348.3,318.5
XS GIS Cut Line= 4
     1911708.241      399968.337     1912041.575      400089.865
     1912116.227      400202.712     1912452.512      400344.032
#Sta/Elev= 30
       0 1749.78    38.4 1735.96      48 1733.34    57.5 1731.97    67.1  1731.1
   153.4 1724.21     163 1723.96   172.6 1724.33     211 1726.57   249.3 1727.57
   287.7 1727.88   354.8  1727.5   393.4 1726.66   403.1 1725.98   412.8 1723.88
   422.4 1720.73   432.1 1719.79   443.5 1721.16   461.1 1723.84   480.4 1725.87
   576.5 1728.96   643.7 1731.55   682.1  1733.4   710.9 1735.13   720.5 1736.22
   749.3 1742.18   806.9 1752.17   826.1 1754.77   845.3 1756.34   854.9 1756.88
#Mann= 3 , 0 , 0
       0      .1       0   422.4    .045       0   443.5      .1       0
Bank Sta=422.4,443.5
XS Rating Curve= 0 ,0
Exp/Cntr=0.3,0.1

Type RM Length L Ch R = 1 ,11360.3 ,77.9,69,59.8
XS GIS Cut Line= 4
       1911567.1      400293.518     1911768.923      400332.581
     1911890.451      400308.709     1912276.735      400384.664
#Sta/Elev= 30
       0 1739.17     9.8 1735.89    39.2 1726.86    48.9 1724.63    58.7 1723.48
    97.9 1721.44   127.3 1720.25   224.6 1717.13   234.2  1716.4   253.2 1713.65
   262.7 1712.98   272.3 1713.17   273.7 1713.31   281.8 1714.14   291.3 1715.56
   300.8 1716.67   329.4  1718.1   349.1 1719.41   358.9 1719.77   378.6 1719.87
   408.2 1720.33   467.2 1721.76   545.9 1723.27   575.5 1724.09   595.2 1724.81
     605 1725.36   654.2 1728.95   703.4 1732.25   713.3 1733.32   723.1 1735.29
#Mann= 3 , 0 , 0
       0      .1       0   253.2    .045       0   273.7     .06       0
Bank Sta=253.2,273.7
XS Rating Curve= 0 ,0
Exp/Cntr=0.3,0.1

Type RM Length L Ch R = 1 ,11291.2 ,388.7,417,445.3
XS GIS Cut Line= 4
     1911546.093      400390.306     1911799.999      400415.046
     1911896.353      400359.056      1912270.22      400482.921
#Sta/Elev= 30
       0  1743.9     9.8 1741.06    49.1 1728.24    58.9 1725.33    68.7 1723.64
    78.5 1723.04     157 1720.22   215.9 1717.41   245.3 1717.16   292.3 1716.01
   308.4 1713.19   310.8 1712.72   320.1 1711.75   329.4  1712.6     348 1718.95
   357.3 1720.05   366.6  1720.1   385.8 1719.52   433.8 1719.29   462.6 1718.84
   510.6 1719.38   587.5 1721.35   616.3 1721.82   645.1 1724.17   693.2 1726.14
   712.4 1727.96     722 1729.69   731.6 1732.06   750.8 1737.54   760.4    1740
#Mann= 3 , 0 , 0
       0      .1       0   308.4    .045       0   329.4     .08       0
Bank Sta=308.4,329.4
XS Rating Curve= 0 ,0
Exp/Cntr=0.3,0.1

Type RM Length L Ch R = 1 ,10874.2 ,394.6,396.6,398.3
XS GIS Cut Line= 4
     1911491.839      400619.907      1911667.79      400730.317
      1911750.52      400784.838      1912063.02      400866.435
#Sta/Elev= 30
       0 1747.34     9.4 1745.37    18.9 1742.43    56.6 1726.78    66.1 1723.39
    75.5 1720.62    94.4 1715.72   113.3 1710.96   122.8 1708.89   132.2 1707.96
   141.6 1707.75   216.7 1708.28   225.7 1707.68   234.7 1705.65   247.7 1701.32
   252.8 1699.83   261.8 1699.91   267.7 1701.47   270.8 1702.29   279.8 1705.52
   288.8 1707.67   316.6 1708.78   375.3 1712.16   414.5 1714.03   522.1 1717.58
   551.5 1719.14   561.3 1720.18   571.1  1721.8   610.2 1729.97   629.8 1733.33
#Mann= 3 , 0 , 0
       0      .1       0   247.7    .045       0   267.7      .1       0
Bank Sta=247.7,267.7
XS Rating Curve= 0 ,0
Exp/Cntr=0.3,0.1

Type RM Length L Ch R = 1 ,10477.6 ,473.4,479.3,485.1
XS GIS Cut Line= 4
     1911260.937      400854.282     1911372.304      400986.914
     1911464.318      401058.094     1911755.728      401177.199
#Sta/Elev= 30
       0  1725.4    19.2 1721.24    28.9 1719.57    38.5 1718.45    57.7 1717.24
    86.6 1715.01   105.8 1713.98   125.1 1713.15   153.9 1711.46   163.6 1710.72
   182.9 1708.76   192.6 1707.23   202.3 1703.99     212 1698.92   220.7 1695.47
   221.7 1695.07   231.4 1694.21   240.7 1695.83   250.7 1698.12   260.4 1699.62
   328.9 1702.23   348.6 1702.49   387.9  1702.4   397.7 1702.64   446.9 1704.93
     506 1708.49   555.1 1710.19     565 1710.78   584.6 1712.41   604.3 1713.56
#Mann= 3 , 0 , 0
       0      .1       0   220.7    .045       0   240.7      .1       0
Bank Sta=220.7,240.7
XS Rating Curve= 0 ,0
Exp/Cntr=0.3,0.1

Type RM Length L Ch R = 1 ,9998.4  ,406.6,392.7,378.4
XS GIS Cut Line= 3
      1911038.97      401115.386     1911167.443      401271.636
     1911341.054      401476.497
#Sta/Elev= 30
       0 1723.65     9.6 1720.75    19.3 1718.17    28.9 1716.19    67.4 1709.04
     106 1702.18   115.6 1699.57   125.2 1695.28   134.9 1690.42   144.5 1688.19
   154.1 1689.05   163.8 1691.44   173.4 1693.86     183 1694.95   192.6 1695.51
   269.4 1698.74     279 1699.04   307.8 1699.58   317.4 1699.91     327 1700.71
   346.1 1703.85   365.3 1706.73   374.9  1708.3   384.5 1710.26   394.1 1712.55
   422.9 1720.32   432.4 1722.72     442 1724.88   451.6 1726.83   470.8 1730.22
#Mann= 3 , 0 , 0
       0      .1       0   134.9    .045       0   163.8      .1       0
Bank Sta=134.9,163.8
XS Rating Curve= 0 ,0
Exp/Cntr=0.3,0.1

Type RM Length L Ch R = 1 ,9605.7  ,155.3,169.4,181.9
XS GIS Cut Line= 4
     1910714.318      401424.414     1910847.998      401514.692
     1910943.484      401545.942     1911089.318      401641.428
#Sta/Elev= 29
       0 1717.56      38 1707.89    47.4 1705.62    56.9 1703.39    75.9 1699.16
    85.4 1697.26    94.9 1695.79   104.4 1694.91   161.3 1691.26   170.4 1690.58
   179.6 1688.96   197.2 1683.45   197.8 1683.26     207 1682.06   216.1 1683.53
   217.2 1683.99   225.2 1687.33   234.4 1690.35   243.5 1691.35   261.8 1692.65
   300.5 1695.03   310.2 1695.55   329.6 1696.32   339.2 1697.01   348.9 1698.23
   358.6 1700.34   397.4 1709.52   416.7 1713.78   436.1 1717.73
#Mann= 3 , 0 , 0
       0      .1       0   197.2    .045       0   217.2      .1       0
Bank Sta=197.2,217.2
XS Rating Curve= 0 ,0
Exp/Cntr=0.3,0.1

Type RM Length L Ch R = 1 ,9436.2  ,166.3,155.3,144.7
XS GIS Cut Line= 3
     1910701.996      401512.181      1910860.85      401703.588
     1911000.173      401716.608
#Sta/Elev= 27
       0 1703.84    19.1 1699.52    38.3 1695.55    47.8 1693.76    57.4 1692.37
      67 1691.53    86.1 1690.15   105.2 1688.66   114.8    1688   124.4 1687.44
   153.1 1686.15   191.3 1684.74   200.9 1683.97   213.8 1682.17     220 1681.33
   229.6 1681.33   233.8  1682.2   239.2 1683.33   248.7  1685.9   258.1 1687.46
     286 1690.16   295.4 1691.53   323.4 1696.94     342 1700.37   360.7 1703.57
   379.3 1706.67   388.7 1708.16
#Mann= 3 , 0 , 0
       0      .1       0   213.8    .045       0   233.8      .1       0
Bank Sta=213.8,233.8
XS Rating Curve= 0 ,0
Exp/Cntr=0.3,0.1

Type RM Length L Ch R = 1 ,9280.9  ,443.9,436.7,429.5
XS GIS Cut Line= 4
      1910538.97      401655.317     1910665.707      401703.928
     1910750.776      401742.122     1911012.929      401752.539
#Sta/Elev= 30
       0 1723.26     9.7 1722.49    19.4 1721.13    29.1 1719.16    38.8 1716.43
    48.5 1712.85    58.2 1708.85    87.3 1696.81   106.6 1688.16   116.4 1684.36
     126  1681.7   135.7 1680.46   145.1 1679.86   154.4 1678.55   163.7  1676.1
     173 1675.02   182.4  1676.1   186.6 1677.85     201 1683.92   210.3 1685.22
   316.4 1687.57   335.9 1688.33     365 1690.13   374.7 1691.22   384.5 1693.45
   394.2 1696.07   403.9 1698.04   413.6 1699.53   442.8 1703.03   491.4 1708.04
#Mann= 3 , 0 , 0
       0      .1       0   163.7    .045       0   186.6      .1       0
Bank Sta=163.7,186.6
XS Rating Curve= 0 ,0
Exp/Cntr=0.3,0.1

Type RM Length L Ch R = 1 ,8844.2  ,252.1,301.2,348
XS GIS Cut Line= 3
     1910554.595      401963.476     1910797.651      402123.198
     1911000.776       402149.24
#Sta/Elev= 30
       0  1702.1     9.7 1700.09    19.4  1697.7    38.8 1692.59    48.5 1689.73
    67.9 1683.28    77.6 1680.62    87.2 1679.15      97 1678.48     126 1677.55
   155.1 1676.82   193.9 1676.09   213.3 1675.83   232.7 1675.71   300.6  1675.8
   310.3  1674.8   319.4 1672.44   329.8 1669.82   339.4 1669.77   344.11671.476
   349.4  1673.4   359.1  1679.1   368.8 1683.67   388.4 1690.65   398.1  1693.8
   407.9 1696.25   417.6 1698.43   437.1 1702.62   476.1 1710.58   495.6 1714.17
#Mann= 3 , 0 , 0
       0      .1       0   319.4    .045       0   344.1      .1       0
Bank Sta=319.4,344.1
XS Rating Curve= 0 ,0
Exp/Cntr=0.3,0.1

Type RM Length L Ch R = 1 ,8543    ,279.5,253.6,228.4
XS GIS Cut Line= 4
     1910565.012       402015.56     1910626.605      402203.674
     1910574.522      402319.777     1910767.664      402490.133
#Sta/Elev= 30
       0 1693.86    18.8 1690.01    28.3 1687.72    56.6 1679.69      66 1677.45
    75.4 1675.78    84.8 1674.53    94.3 1673.48   103.7 1672.53   113.1  1671.8
     132  1670.9   160.2 1669.96   188.5 1669.47   237.1 1669.48   246.9 1669.24
   256.7 1668.57   273.6 1666.18   276.2 1665.79     286 1665.28   295.8 1666.73
   305.6 1669.91   315.4 1672.77   325.2 1673.45   334.7 1673.88   372.9 1674.63
   458.7 1675.83     516 1678.49     535 1679.51   573.2 1682.01   582.7 1683.06
#Mann= 3 , 0 , 0
       0      .1       0   273.6    .045       0   295.8      .1       0
Bank Sta=273.6,295.8
XS Rating Curve= 0 ,0
Exp/Cntr=0.3,0.1

Type RM Length L Ch R = 1 ,8289.4  ,109.2,112,114.9
XS GIS Cut Line= 5
     1910458.159       401888.57     1910469.526      402045.073
     1910417.443      402147.504      1910476.47      402236.046
      1910592.79       402617.99
#Sta/Elev= 30
       0 1707.22    19.6 1704.69    29.4 1703.82    78.5 1700.55    98.1 1698.87
   137.3 1695.13   156.9 1692.73   166.5 1690.98   204.8 1683.03   262.2 1672.64
   291.2 1667.66   300.8 1665.25   310.5 1662.13   320.2 1659.78   329.9 1659.55
   339.6 1661.16   349.2 1663.07   358.9 1663.83   407.5 1664.26   426.9 1664.87
   465.9 1667.23   495.1 1670.47   504.8 1670.84   524.3 1670.42   592.5 1667.81
   602.2 1667.66     612 1668.11   689.9 1676.62   748.3 1684.12   777.5 1688.38
#Mann= 3 , 0 , 0
       0      .1       0   310.5    .045       0   339.6      .1       0
Bank Sta=310.5,339.6
XS Rating Curve= 0 ,0
Exp/Cntr=0.3,0.1

Type RM Length L Ch R = 1 ,8177.4  ,306.8,304.1,301
XS GIS Cut Line= 4
     1910080.555      401918.952     1910295.915      402144.032
     1910375.694      402296.556     1910526.818      402673.546
#Sta/Elev= 30
       0 1701.32    38.9 1698.09    68.1  1695.1    77.9 1693.54   116.8 1685.88
   155.8    1679   175.2 1675.93     185 1674.96   204.4 1674.01   311.5  1670.9
   321.1 1670.12   359.3 1664.92   378.4 1662.86  410.45 1657.16   416.7 1656.34
   426.3 1656.03   435.8  1656.3   445.4 1657.67     455 1661.03   464.5 1662.57
   570.7 1664.14   609.4 1667.32     619 1667.08   667.4 1664.28     677 1664.06
   686.7 1664.56   696.4 1665.74   754.4 1674.57   812.4 1682.52   889.8 1694.88
#Mann= 3 , 0 , 0
       0      .1       0  410.45    .045       0   445.4      .1       0
Bank Sta=410.45,445.4
XS Rating Curve= 0 ,0
Exp/Cntr=0.3,0.1

Type RM Length L Ch R = 1 ,7873.4  ,312.4,300.5,288.4
XS GIS Cut Line= 3
     1909951.258      402170.833     1910097.091      402386.111
     1910241.188      402665.625
#Sta/Elev= 30
       0 1683.21     9.6 1682.31    19.3 1681.02    57.8 1675.01      77 1672.53
   144.5  1665.5     183 1662.13   192.6 1660.39   202.2 1657.31   211.9 1655.11
   221.5 1654.81   231.1 1656.22   240.8 1658.31   250.4 1659.01     319 1658.33
   348.5 1658.52   358.3 1658.43     378 1657.85   387.8 1657.75   397.6 1658.01
   417.3 1659.53   446.7 1662.41   456.6 1663.86   466.4 1666.06   515.5 1678.55
   525.4 1681.16   535.2  1684.2   554.8 1690.67   564.7 1692.73   574.5 1693.04
#Mann= 3 , 0 , 0
       0      .1       0   202.2    .045       0   231.1      .1       0
#XS Ineff= 2 , 0
                          276.44         1660.66
Permanent Ineff=
       F       F
Bank Sta=202.2,231.1
XS Rating Curve= 0 ,0
Exp/Cntr=0.3,0.1

Type RM Length L Ch R = 1 ,7572.8  ,206.6,206.6,206.6
XS GIS Cut Line= 4
     1909666.536       402314.93     1909803.254      402504.817
      1910002.43      402613.397     1910082.725      402689.352
#Sta/Elev= 30
       0 1688.21    58.5 1682.03    87.7 1678.68    97.5  1677.5     117 1674.91
   136.5 1671.64   165.7 1668.19   175.5 1666.92   204.7 1662.82   214.5 1661.72
     234 1660.08   243.4 1658.77   252.9 1656.21   261.2 1653.55   262.3  1653.2
   271.8 1651.75   281.2 1653.19   290.7 1655.74   300.2 1657.02   309.6 1657.38
   385.2 1657.41   413.6 1657.53   432.5 1657.99   460.8 1658.98   497.7 1660.07
   506.9 1660.58   516.1 1661.73   525.3 1663.52   552.9 1669.37   571.4 1673.14
#Mann= 3 , 0 , 0
       0      .1       0   261.2    .045       0   281.2      .1       0
Bank Sta=261.2,281.2
XS Rating Curve= 0 ,0
Exp/Cntr=0.3,0.1

Type RM Length L Ch R = 1 ,7366.2  ,313.2,321.3,329.4
XS GIS Cut Line= 4
     1909574.912      402472.338      1909846.18      402687.181
     1909941.666      402737.095     1909991.579      402782.667
#Sta/Elev= 30
       0 1678.18    38.4 1670.84    67.3 1665.65    76.9  1664.1    86.5 1662.72
    96.1 1661.64   105.7 1660.86   115.4 1660.51     125 1660.32     173 1660.23
   182.6 1660.17   201.9 1659.87   278.8 1658.03   307.6 1657.08     346 1655.46
   365.6 1654.79   375.4 1653.91   385.2 1651.88   392.3 1650.23     395  1649.6
   404.8  1648.7   414.6 1650.12   424.4 1653.63   434.2 1656.93   453.8 1658.57
   463.4 1659.93   473.1 1661.74   482.8  1663.9   511.7  1671.3   521.4 1673.57
#Mann= 3 , 0 , 0
       0      .1       0   392.3    .045       0   414.6      .1       0
Bank Sta=392.3,414.6
XS Rating Curve= 0 ,0
Exp/Cntr=0.3,0.1

Type RM Length L Ch R = 1 ,7044.9  ,183.2,167.6,151.9
XS GIS Cut Line= 5
     1909242.707      402478.125     1909506.965      402694.439
     1909594.526      402792.469     1909679.595      402881.011
      1909882.72      402886.219
#Sta/Elev= 30
       0 1684.43    48.8 1680.64    68.3 1678.47   117.1  1672.4   126.8 1671.48
   185.4 1666.92   234.2 1664.28   273.2 1661.95     322  1660.6   341.5 1659.61
   360.3 1658.26   369.7 1657.86   435.4 1655.94   454.2 1655.16   482.4 1653.38
   491.8 1652.37   501.3 1650.33   510.7 1648.36   520.2 1647.94   529.6 1649.66
   539.1 1651.61   548.5  1652.6   624.8 1655.25   644.1 1656.63   653.8  1657.1
   673.1 1657.02   711.8 1660.59   750.5  1663.5   769.9 1664.62   798.9 1665.92
#Mann= 3 , 0 , 0
       0      .1       0   501.3    .045       0   529.6      .1       0
Bank Sta=501.3,529.6
XS Rating Curve= 0 ,0
Exp/Cntr=0.3,0.1

Type RM Length L Ch R = 1 ,6877.3  ,271.1,242.6,214.1
XS GIS Cut Line= 4
     1909013.541         403025.     1909438.276      402950.455
     1909617.095      402983.442     1909828.901      402910.525
#Sta/Elev= 30
       0 1719.33    29.4 1715.94    39.2  1714.6    68.6 1709.84      98 1705.61
   137.2 1700.22   176.4 1695.23     196 1691.13   215.6 1687.44   225.4 1685.85
   254.8 1681.68   303.8 1674.21   421.4 1658.12   431.2 1656.48   450.4 1652.69
   459.9 1651.19   469.5 1650.31   526.9 1647.12   536.5 1646.67   546.1 1646.65
   555.6 1647.75   565.2    1650   574.8  1651.8   603.5 1653.77   622.8 1654.62
   642.3  1655.1   700.7 1655.52   749.4 1657.11   788.4  1659.2   837.1 1662.61
#Mann= 3 , 0 , 0
       0      .1       0   526.9    .045       0   555.6      .1       0
Bank Sta=526.9,555.6
XS Rating Curve= 0 ,0
Exp/Cntr=0.3,0.1

Type RM Length L Ch R = 1 ,6634.7  ,332,317.9,303.8
XS GIS Cut Line= 5
     1909419.179      403356.705     1909575.429      403229.969
     1909627.512      403157.053     1909676.123      403042.469
     1909863.623      402950.455
#Sta/Elev= 30
       0 1695.76    57.5 1686.38   124.5 1675.11   134.1 1673.33   143.7 1671.23
   153.3 1668.53   162.9 1666.22   172.4 1664.63   191.6 1662.42   201.2 1661.17
   210.2 1658.79   219.1 1654.37   228.1 1649.25     237 1647.15     246 1647.46
     255 1648.99   263.9 1650.28   272.9 1650.66   300.4 1650.47   348.2 1650.54
     377 1649.68   386.5 1649.26   396.1 1649.28   415.3 1650.64   443.7 1651.44
   453.2 1651.94   481.7 1654.35   500.7 1655.63   576.7  1659.6   624.1 1662.36
#Mann= 3 , 0 , 0
       0      .1       0   228.1    .045       0     255      .1       0
#XS Ineff= 2 , 0
                          360.38         1652.79
Permanent Ineff=
       F       F
Bank Sta=228.1,255
XS Rating Curve= 0 ,0
Exp/Cntr=0.3,0.1

Type RM Length L Ch R = 1 ,6316.7  ,202.5,216,229.4
XS GIS Cut Line= 4
      1909788.97      403415.733     1909828.901      403127.539
     1909837.582      403012.955     1909879.248      402952.192
#Sta/Elev= 30
       0 1672.64    38.8 1669.73    58.2 1667.84    77.6 1665.34   126.1  1657.7
   135.8 1656.45   155.2 1654.49   164.9 1653.93   174.6 1653.75   203.7 1654.28
   232.8 1654.45   242.5  1654.3   252.2  1653.8   300.5 1649.78   310.1 1647.83
   319.7 1644.36   329.2 1642.49   338.8 1643.58   341.5 1644.66   348.4 1647.43
     358 1650.29   367.6 1650.85   377.1 1650.64   386.7 1650.83   396.3 1651.99
   405.9 1653.94   433.5 1659.02   442.7  1660.3   461.1 1661.93   479.5 1663.01
#Mann= 3 , 0 , 0
       0      .1       0   319.7    .045       0   341.5      .1       0
Bank Sta=319.7,341.5
XS Rating Curve= 0 ,0
Exp/Cntr=0.3,0.1

Type RM Length L Ch R = 1 ,6100.7  ,372.6,383.5,393.5
XS GIS Cut Line= 2
     1909853.207      403405.317     1910117.095      403025.108
#Sta/Elev= 30
       0 1666.48    19.3 1665.41    28.9 1664.69    38.6 1663.27    48.2 1661.55
    67.5 1657.79    77.1 1656.38    86.8 1655.63   144.6 1652.59   173.6 1651.24
   212.1 1649.86   260.3 1648.47     270 1648.09   279.6 1647.52   289.3 1645.53
   298.9 1641.55   308.5 1639.11   318.2  1639.8   320.3 1640.49   327.8 1642.94
   337.5  1646.6   347.1 1649.45   366.4 1654.62     376  1656.9   385.7 1658.85
   395.3 1661.21   414.6 1666.39   424.2 1668.28   433.9 1669.73   462.8  1673.4
#Mann= 3 , 0 , 0
       0      .1       0   298.9    .045       0   320.3      .1       0
Bank Sta=298.9,320.3
XS Rating Curve= 0 ,0
Exp/Cntr=0.3,0.1

Type RM Length L Ch R = 1 ,5717.2  ,263.9,263.7,265.5
XS GIS Cut Line= 3
      1910007.72      403574.587     1910235.151      403432.226
     1910358.415      403307.226
#Sta/Elev= 27
       0 1664.04    28.8 1659.42    57.5  1655.3    95.8    1650     115 1647.14
   124.6 1645.86   134.2 1645.06   143.7 1644.74   153.3  1644.3   162.9 1643.76
   191.6 1641.88   201.2 1639.71   210.8  1634.8     219 1631.39   220.4 1630.81
     230 1629.61   239.6 1631.38   249.2 1634.91   258.7 1637.05   268.3 1637.99
   297.6 1640.56   326.8 1643.31   356.1 1646.35   365.8 1647.44   414.6 1653.31
   434.1 1656.21   443.9 1657.56
#Mann= 3 , 0 , 0
       0      .1       0     219    .045       0   239.6      .1       0
Bank Sta=219,239.6
XS Rating Curve= 0 ,0
Exp/Cntr=0.3,0.1

Type RM Length L Ch R = 1 ,5453.5  ,152.7,179.6,203.1
XS GIS Cut Line= 4
     1910051.123      403591.948     1910370.568      403642.296
     1910450.429      403572.851     1910620.568      403442.643
#Sta/Elev= 30
       0 1656.41    39.2 1648.98    58.8 1646.61      98 1644.48   107.8 1645.32
   127.4 1648.46     147 1649.08   166.6 1647.28   205.8 1641.22   235.2 1638.62
   254.8 1637.57     294 1637.26   323.4 1636.13     333 1634.89   352.2 1629.54
   361.9 1628.41   371.5 1628.62   381.1 1630.15   400.4  1633.7     410 1634.89
   419.6 1635.93   448.7 1637.25   458.4 1638.86   468.2 1641.04   487.6 1646.92
   526.6 1661.07   546.1 1665.94   594.8 1674.95     624 1677.72   643.5 1680.19
#Mann= 3 , 0 , 0
       0      .1       0   352.2    .045       0   381.1      .1       0
Bank Sta=352.2,381.1
XS Rating Curve= 0 ,0
Exp/Cntr=0.3,0.1

Type RM Length L Ch R = 1 ,5274    ,613.7,611,608.1
XS GIS Cut Line= 4
     1910063.276      403652.365     1910407.026      403706.532
     1910535.498      403770.768     1910721.262      403883.615
#Sta/Elev= 30
       0 1654.87      29 1648.55    38.7 1647.16    48.3 1646.39    77.3  1644.6
   125.7 1642.27   154.7 1641.63   164.3 1641.23     174 1640.57   222.3 1635.85
     232 1635.26   299.7 1634.53   338.3 1634.48   357.6  1634.2   367.1  1633.6
   376.7 1631.94   394.1 1626.87   395.9 1626.37   405.4 1625.51     415 1626.79
   434.2 1632.23   443.8  1634.5   453.3 1636.22   462.9 1637.32   501.1 1640.66
   595.6  1647.4   642.8 1650.23   652.3 1651.27   661.7 1653.44     709 1667.87
#Mann= 3 , 0 , 0
       0      .1       0   394.1    .045       0     415      .1       0
Bank Sta=394.1,415
XS Rating Curve= 0 ,0
Exp/Cntr=0.3,0.1

Type RM Length L Ch R = 1 ,4662.9  ,153.4,150.2,147.1
XS GIS Cut Line= 4
     1910005.984       404171.81     1910184.804      404249.935
     1910275.082      404282.921     1910542.443      404310.698
#Sta/Elev= 30
       0  1655.1     9.8 1653.75    29.3 1650.77    58.5 1645.92   117.1 1635.36
   146.4 1629.82   185.4 1623.23   195.1 1621.48   204.8 1619.17   214.4 1616.37
     224 1614.22   233.6 1614.69   236.9 1615.45   243.2  1616.9   252.8 1618.91
   262.4 1619.83   281.6 1621.24   291.3 1621.66   300.9 1622.34   310.5 1623.12
   339.3 1625.72   377.7 1628.88   387.3 1629.49   396.9 1629.93   444.9 1631.54
   464.1 1632.39   512.1 1634.08   521.7 1634.52   540.9 1635.82   560.1 1637.59
#Mann= 3 , 0 , 0
       0      .1       0   214.4    .045       0   236.9      .1       0
Bank Sta=214.4,236.9
XS Rating Curve= 0 ,0
Exp/Cntr=0.3,0.1

Type RM Length L Ch R = 1 ,4512.7  ,104.7,97.9,90.9
XS GIS Cut Line= 4
     1909919.179      404266.428     1910104.943      404387.955
     1910233.415      404417.469     1910535.498       404434.83
#Sta/Elev= 30
       0 1652.55    67.6 1648.87    96.5  1647.4   106.2 1647.24   115.8 1647.44
   125.5 1647.36   135.1 1646.08   144.8 1642.79   164.1 1634.97   173.7 1631.29
     193 1624.55   212.3 1616.54     222 1613.47   231.4  1612.3   240.8 1611.55
   259.6 1610.29   269.1 1609.52   278.5 1608.95   287.9 1608.84   297.3 1609.38
   316.1 1612.06   325.6 1612.91     335 1613.47   353.8 1614.17   373.3 1615.14
   461.2 1620.34   490.4 1622.16   578.3 1628.84   607.6 1631.22   656.4 1634.86
#Mann= 3 , 0 , 0
       0      .1       0   269.1    .045       0   297.3      .1       0
Bank Sta=269.1,297.3
XS Rating Curve= 0 ,0
Exp/Cntr=0.3,0.1

Type RM Length L Ch R = 1 ,4414.8  ,259.1,240.9,221.5
XS GIS Cut Line= 4
     1909900.082      404636.219     1910111.887      404500.803
     1910216.054      404495.594     1910519.873      404545.942
#Sta/Elev= 30
       0 1647.12     9.7 1647.58      29 1649.71    38.7 1650.33    48.4 1650.11
   135.4 1645.33   154.7 1645.18   164.4 1644.73     174 1643.64   183.7 1642.16
   193.4  1640.3     203  1638.2   212.7 1635.34   232.1 1628.94   260.9 1620.06
   270.4 1616.85   279.8 1612.95   289.3 1608.71   298.8 1606.38   308.3 1606.63
   317.8 1607.57   346.2 1610.01   374.9 1611.55   403.8 1612.45   471.2 1613.39
   490.4 1613.98   528.9 1616.78   557.8 1619.23   644.4 1628.27   663.6 1629.95
#Mann= 3 , 0 , 0
       0      .1       0   289.3    .045       0   317.8     .07       0
Bank Sta=289.3,317.8
XS Rating Curve= 0 ,0
Exp/Cntr=0.3,0.1

Type RM Length L Ch R = 1 ,4173.8  ,475.1,496.6,518.1
XS GIS Cut Line= 4
     1910058.068      404799.414     1910242.095      404726.497
     1910365.359      404601.497     1910518.137      404604.969
#Sta/Elev= 30
       0 1658.22     9.4 1657.31    18.8 1655.99    56.6  1648.6    75.4    1644
    94.3 1638.47   103.7 1635.21   113.1 1631.31   150.8 1614.21   160.2 1609.51
   169.7 1605.07   179.1 1602.43   188.5    1602     198 1602.52   207.7 1602.79
   217.4  1602.8     237 1602.17   256.5 1600.82   266.2 1600.35     276 1600.25
   285.7 1600.77   295.5  1602.4   305.2 1604.35   324.7  1607.8     354 1612.79
   363.8 1614.08     383 1615.47   421.3 1617.84   459.5 1620.61   526.3 1626.92
#Mann= 3 , 0 , 0
       0      .1       0   256.5    .045       0   285.7      .1       0
#XS Ineff= 2 , 0
          213.61 1604.59
Permanent Ineff=
       F       F
Bank Sta=256.5,285.7
XS Rating Curve= 0 ,0
Exp/Cntr=0.3,0.1

Type RM Length L Ch R = 1 ,3677.2  ,523.7,526.6,529
XS GIS Cut Line= 3
      1910124.04      405080.664      1910320.22       405091.08
     1910479.943      405065.039
#Sta/Elev= 24
       0  1644.7    29.5 1638.16    49.1 1633.62    58.9 1631.26    68.8 1628.61
    78.6 1625.31    88.4 1620.94    98.2  1615.4     108 1609.19   117.9 1602.64
   127.7 1595.23   137.5 1586.11   147.3 1577.25  154.421574.416   157.2 1573.31
     167 1574.07   179.3 1576.07   186.6 1577.37   196.5 1578.95     225  1583.7
   272.6 1591.84   310.7 1597.66   320.2 1599.19   358.3 1605.59
#Mann= 3 , 0 , 0
       0      .1       0  154.42    .045       0   179.3      .1       0
Bank Sta=154.42,179.3
XS Rating Curve= 0 ,0
Exp/Cntr=0.3,0.1

Type RM Length L Ch R = 1 ,3150.6  ,505.5,493.5,481.4
XS GIS Cut Line= 3
     1910131.635      405574.804     1910353.858      405611.263
     1910510.108      405597.374
#Sta/Elev= 30
       0 1576.19    29.4 1567.32      49 1561.54    58.8 1558.74    68.5  1556.3
    78.3 1554.72    88.1 1553.76    97.9 1553.01   117.5 1551.82   146.9 1550.37
   156.7 1549.64   166.4 1548.23   176.2 1545.84     186 1544.04   195.8 1545.59
   196.7 1545.92   205.6 1549.17   215.4 1552.35   244.8  1559.1   254.6 1561.55
   264.4 1564.16     284 1569.62   293.8 1572.22   303.6 1574.64   313.4 1576.95
     333 1581.36   342.8 1583.33   352.6 1585.03   362.4 1586.49   382.1 1589.18
#Mann= 3 , 0 , 0
       0      .1       0   176.2    .045       0   196.7      .1       0
Bank Sta=176.2,196.7
XS Rating Curve= 0 ,0
Exp/Cntr=0.3,0.1

Type RM Length L Ch R = 1 ,2657    ,246.9,244.9,242.8
XS GIS Cut Line= 3
     1910004.248      406131.011     1910216.054      406061.567
      1910320.22       405966.08
#Sta/Elev= 28
       0 1566.38    19.4 1559.43    29.1 1555.84    77.5 1537.68   116.3 1523.82
     126 1520.59   135.7 1517.83   145.4 1515.52   164.8 1511.47   173.8 1509.71
   174.4 1509.59   184.1 1508.59   193.8 1509.54   203.5 1512.97   213.2 1517.44
   222.9 1521.62   241.7 1530.23   251.2 1533.76   260.6 1536.54     270 1539.06
   279.4 1541.29   288.8 1543.19   298.3 1544.74   307.7 1545.76   317.1 1546.52
   326.5 1547.14   354.8 1548.37   364.2 1548.68
#Mann= 3 , 0 , 0
       0      .1       0   173.8    .045       0   193.8      .1       0
Bank Sta=173.8,193.8
XS Rating Curve= 0 ,0
Exp/Cntr=0.3,0.1

Type RM Length L Ch R = 1 ,2412.1  ,195.8,186.9,177.4
XS GIS Cut Line= 4
     1910091.232       406360.72     1910247.482      406306.901
     1910309.982      406280.859     1910421.093      406187.109
#Sta/Elev= 30
       0 1556.09    19.4 1545.74    29.2 1540.67    38.9 1535.72    48.6 1530.88
    58.3 1526.25      68 1521.96    87.5 1514.42    97.2    1510   106.9 1505.75
   116.6  1503.5   126.4 1502.69   136.1 1502.02   165.3 1500.31   174.9 1499.42
   184.6 1497.84   192.5 1496.25   194.3 1495.89     204 1494.99   213.6 1496.53
   223.3 1499.12     233 1500.77   242.7  1501.8   271.7 1504.57   291.1 1506.65
   310.5 1508.84   329.9  1511.2   349.3 1513.76   368.6 1516.59   378.4 1518.23
#Mann= 3 , 0 , 0
       0      .1       0   192.5    .045       0   213.6      .1       0
Bank Sta=192.5,213.6
XS Rating Curve= 0 ,0
Exp/Cntr=0.3,0.1

Type RM Length L Ch R = 1 ,2225.2  ,461,464.9,468.5
XS GIS Cut Line= 2
      1910217.79      406598.025      1910507.72      406320.247
#Sta/Elev= 30
       0 1541.25     9.8 1535.06    19.6 1529.43    29.4  1524.7    39.2 1520.36
      49 1516.57    58.8  1513.6    68.6 1510.98    88.1 1506.12    97.9 1503.85
   117.5 1499.61   166.5  1489.5   176.3 1486.89   186.1 1483.47   193.9 1481.37
   195.9 1480.83   205.7 1481.16   215.4 1484.13   225.2 1487.32     235 1489.75
   264.4 1495.99   274.2 1497.84     284 1498.76   293.8 1499.31   323.2 1500.69
     333 1501.29   342.8 1502.04   381.9 1505.31   391.7 1506.37   401.5 1508.09
#Mann= 3 , 0 , 0
       0      .1       0   193.9    .045       0   215.4      .1       0
Bank Sta=193.9,215.4
XS Rating Curve= 0 ,0
Exp/Cntr=0.3,0.1

Type RM Length L Ch R = 1 ,1760.4  ,286.8,299.1,311.7
XS GIS Cut Line= 3
     1910464.318      406940.907     1910636.193      406819.379
     1910731.679      406722.157
#Sta/Elev= 27
       0 1513.58    19.1 1506.72    28.7 1503.15    38.3 1499.46    57.4 1491.68
      67  1487.5    76.6 1483.09    86.1 1478.35    95.7 1473.37   105.2 1468.22
   124.4 1457.12     134 1453.09   143.5 1451.73   153.1 1452.31   159.4 1453.11
   162.7 1453.53   181.8 1456.41   191.4 1457.74   200.9 1459.22   210.5 1460.87
   239.7 1466.62   259.2 1470.66   288.4 1476.94   307.8 1481.26   317.6 1483.36
   327.3 1485.28   346.8  1488.7
#Mann= 3 , 0 , 0
       0      .1       0     134    .045       0   159.4      .1       0
Bank Sta=134,159.4
XS Rating Curve= 0 ,0
Exp/Cntr=0.3,0.1

Type RM Length L Ch R = 1 ,1461.2  ,237,243.6,249.4
XS GIS Cut Line= 4
     1910567.327      407063.469      1910766.98      407035.257
     1910834.254      407026.577     1910922.145      406984.259
#Sta/Elev= 30
       0 1474.41     9.6 1469.32    19.2 1465.16    38.4 1456.49      48 1452.54
    57.6 1449.24    67.2 1446.73    76.8 1445.07    86.4  1444.1      96 1443.61
   105.6 1443.87   115.2 1444.48     144 1445.58   172.8 1446.85     192 1447.26
   201.6 1447.27   211.3 1447.01     221 1446.17   230.5 1444.79   240.4 1443.31
   250.1  1443.8   250.5 1443.92   259.8 1446.82   269.5 1451.33   279.2 1455.58
   298.7 1463.34   318.2  1471.7     328 1475.76   347.5 1483.44     367 1490.92
#Mann= 3 , 0 , 0
       0      .1       0   230.5    .045       0   250.5      .1       0
#XS Ineff= 2 , 0
          184.41 1448.26
Permanent Ineff=
       F       F
Bank Sta=230.5,250.5
XS Rating Curve= 0 ,0
Exp/Cntr=0.3,0.1

Type RM Length L Ch R = 1 ,1217.7  ,260,252.5,245.4
XS GIS Cut Line= 4
     1910566.748      407263.823     1910684.804      407251.671
     1910776.818      407262.087     1910959.109      407208.268
#Sta/Elev= 29
       0 1470.33    36.5 1458.72    82.2 1443.97   100.4 1438.08   109.6 1434.92
   118.7 1430.83   127.9  1425.2   137.2 1419.93   143.5 1418.15   146.5  1417.3
   155.7 1417.31     165  1419.2   174.2 1421.96   183.5 1424.55   211.3 1431.83
   239.8 1439.73   249.3 1442.09   258.8 1443.89   268.3 1445.12   287.3 1447.24
   315.8 1450.23   325.3 1451.35   344.3  1453.8   353.8 1455.13   363.3 1456.67
   372.8 1458.73   382.3 1461.48   391.8 1464.81   401.4 1468.36
#Mann= 3 , 0 , 0
       0      .1       0   143.5    .045       0     165      .1       0
Bank Sta=143.5,165
XS Rating Curve= 0 ,0
Exp/Cntr=0.3,0.1

Type RM Length L Ch R = 1 ,965.1   ,266.1,269.8,272.5
XS GIS Cut Line= 3
     1910617.783      407527.879      1910791.81      407496.629
     1910932.887      407444.545
#Sta/Elev= 29
       0 1449.21     9.8  1446.6    19.6 1443.78    29.5 1440.55    39.3 1437.03
    49.1  1433.9    58.9 1431.38    68.8    1429    78.6 1426.45    98.2 1421.15
     108  1418.4   117.9 1415.45   127.7 1412.25   135.9 1410.15   137.5 1409.74
   147.3 1409.22   157.2 1410.72     167 1413.24   176.8 1415.58   186.2 1417.49
   214.4 1422.96   242.6 1428.57     252 1430.24   261.4 1431.63   280.2 1434.19
     299 1436.88   308.4 1438.55   317.8 1440.56   327.2 1442.67
#Mann= 3 , 0 , 0
       0      .1       0   135.9    .045       0   157.2      .1       0
Bank Sta=135.9,157.2
XS Rating Curve= 0 ,0
Exp/Cntr=0.3,0.1
